--- LILAURELFK.prj (project) ---

Proj Title=LILAURELFK
Current Plan=p01
Default Exp/Contr=0,0
English Units
Geom File=g01
Flow File=f01
Plan File=p01
BEGIN DESCRIPTION:
---------- MODELED AS PART OF WVEMD CTP PROGRAM, 2023----------
Stream Name: Little Laurel Fork
Flood Zone:  AFH
Upshur County, WV
HEC-RAS Version: RAS 6.3
Vertical Datum: NAVD88
Projection: NAD 1983 StatePlane West Virginia S FIPS 4702 (US Feet)
Terrain: 1-meter LIDAR (FEMA Region III 3DEP collected 2016-2018)
Land Use: 2019 NLCD
Hydrologic Method:
WV SIR2010-5033 regression equations
Additional Model Notes:
Main stem is LAUFSANDRN
END DESCRIPTION:
DSS Export Rating Curves= 0
DSS Export Rating Curve Sorted= 0
DSS Export Volume Flow Curves= 0
DXF OffsetX= 0
DXF OffsetY= 0
DXF ScaleX= 0
DXF ScaleY= 0

--- LILAURELFK.p01 (plan) ---

Plan Title=Floodplain
Program Version=6.31
Short Identifier=Floodplain
Geom File=g01
Flow File=f01
Subcritical Flow
K Sum by GR= 0
Std Step Tol= 0.01
Critical Tol= 0.01
Num of Std Step Trials= 20
Max Error Tol= 0.3
Flow Tol Ratio= 0.001
Split Flow NTrial= 30
Split Flow Tol= 0.02
Split Flow Ratio= 0.02
Log Output Level= 0
Friction Slope Method= 1
Unsteady Friction Slope Method= 2
Unsteady Bridges Friction Slope Method= 1
Parabolic Critical Depth
Global Vel Dist= 0 , 0 , 0
Global Log Level= 0
CheckData=True
Encroach Param=-1 ,0,0, 0
Mapping Interval=1HOUR
Computation Time Step Use Courant=        0
Computation Time Step Use Time Series=    0
Computation Time Step Count To Double=0
Computation Time Step Max Doubling=0
Computation Time Step Max Halving=0
Computation Time Step Residence Courant=0
Run HTab= 0
Run UNet= 0
Run Sediment= 0
Run PostProcess= 0
Run WQNet= 0
Run RASMapper=-1
UNET Theta= 0
UNET Theta Warmup= 0
UNET ZTol= 0
UNET ZSATol= 0
UNET MxIter= 0
UNET Max Iter WO Improvement= 0
UNET MaxInSteps= 0
UNET DtIC= 0
UNET DtMin= 0
UNET MaxCRTS= 0
UNET WFStab= 0
UNET SFStab= 0
UNET WFX= 1
UNET SFX= 1
UNET Gravity=32.17405
UNET 1D Methodology=Finite Difference
UNET DSS MLevel= 1
UNET Pardiso=0
UNET DZMax Abort= 0
UNET Use Existing IB Tables= 0
UNET Froude Reduction=False
UNET Froude Limit= 0
UNET Froude Power= 0
UNET D1 Cores= 0
UNET WindReference=Eulerian
UNET WindDragFormulation=Hsu (1988)
UNET D2 Coriolis=0
UNET D2 Cores= 0
UNET D2 Theta= 1
UNET D2 Theta Warmup= 1
UNET D2 Z Tol= 0.01
UNET D2 Volume Tol= 0.01
UNET D2 Max Iterations= 20
UNET D2 Equation= 0
UNET D2 RampUpFraction=0.1
UNET D2 TimeSlices= 1
UNET D2 Turbulence Formulation=Non-Conservative (original)
UNET D2 Eddy Viscosity=0.3
UNET D2 Transverse Eddy Viscosity=0.1
UNET D2 Smagorinsky Mixing=0
UNET D2 BCVolumeCheck=0
UNET D2 Cores=0
UNET D2 SolverType=PARDISO (Direct)
UNET D2 Minimum Iterations= 3
UNET D2 Maximum Iterations= 30
UNET D2 Restart Number= 10
UNET D2 Relaxation Coeff=1.3
UNET D2 SOR Precondition Iterations= 10
UNET D2 ILUT Maximum Fill= 8
UNET D2 ILUT Tolerance=1E-08
UNET D2 Convergence Tolerance=0.00001
UNET D1D2 MaxIter= 0
UNET D1D2 ZTol=0.01
UNET D1D2 QTol=0.1
UNET D1D2 MinQTol=1
Write IC File= 0
Write IC File at Fixed DateTime=0
Write IC File at Sim End=0
Echo Input=False
Echo Parameters=False
Echo Output=False
Write Detailed= 0
HDF Write Warmup=0
HDF Write Time Slices=0
HDF Flush=0
HDF Compression= 1
HDF Chunk Size= 1
HDF Spatial Parts= 1
HDF Use Max Rows=0
HDF Fixed Rows= 1
Calibration Method= 0
Calibration Iterations= 20
Calibration Max Change=0.05
Calibration Tolerance=0.2
Calibration Maximum=1.5
Calibration Minimum=0.5
Calibration Optimization Method= 1
WQ AD Non Conservative
WQ ULTIMATE=-1
WQ Max Comp Step=1HOUR
WQ Output Interval=15MIN
WQ Output Selected Increments= 0
WQ Create Restart=0
WQ Fixed Restart=0
WQ System Summary=0
WQ Write To DSS=0
Sorting and Armoring Iterations= 10
XS Update Threshold= 0.02
Bed Roughness Predictor= 0
Hydraulics Update Threshold= 0.02
Energy Slope Method= 1
Volume Change Method= 1
Sediment Retention Method= 0
Sediment TS Multiplier= 1
Warm Up Method= 0
XS Weighting Method= 0
Number of US Weighted Cross Sections= 1
Number of DS Weighted Cross Sections= 1
Upstream XS Weight=0
Main XS Weight=1
Downstream XS Weight=0
Number of DS XS's Weighted with US Boundary= 1
Upstream Boundary Weight= 1
Weight of XSs Associated with US Boundary= 0
Number of US XS's Weighted with DS Boundary= 1
Downstream Boundary Weight= 0.5
Weight of XSs Associated with DS Boundary= 0.5
Percentile Method= 0
Sediment Output Level= 3
Mass or Volume Output= 0
Output Increment Type= 1
Profile and TS Output Increment= 1
Transport Output Increment 1
XS Output Flag= 0
XS Output Increment= 10
Read HDF5 Sediment Hotstart= 0
Sediment Hotstart Type= 0
Write Gradation File= 0
Read Gradation Hotstart= 0
Write HDF5 File= 1
Write Binary Output= 1
Write DSS Sediment File= 0
DSS Sediment Output Type= 1
SV Curve= 0
Specific Gage Flag= 0
Subcell Erosion Methods= 0
Subcell Deposition Methods= 0
Advection Scheme= 1
Matrix Solver= 0
Implicit Weighting Factor= 1
Maximum Outer Loop Convergence Iterations= 5
Convergence Maximum Absolute= 0.001
Convergence RMSE= 0.0001
Grain Fractions Max Abs Error= 0.001
Max Subgrid Regions= 1
Max Subgrid Length Scale= 3.402823E+38
Initial Layer Thickness= 3.402823E+38
Min Layer Thickness= 3.402823E+38
Max Layer Thickness= 3.402823E+38
Number of Layers= 5

--- LILAURELFK.f01 (steady flow) ---

Flow Title=Flows
Program Version=6.31
Number of Profiles= 1
Profile Names=01pct
River Rch & RM=LILAURELFK,Main            ,17962
     337
River Rch & RM=LILAURELFK,Main            ,16198
     377
River Rch & RM=LILAURELFK,Main            ,15008
     420
River Rch & RM=LILAURELFK,Main            ,12339
     477
River Rch & RM=LILAURELFK,Main            ,8964
     530
River Rch & RM=LILAURELFK,Main            ,4353
     657
Boundary for River Rch & Prof#=LILAURELFK,Main            , 1
Up Type= 0
Dn Type= 3
Dn Slope=0.04016
DSS Import GetInterval= 0
DSS Import GetPeak= 0
DSS Import FillOption= 0

--- LILAURELFK.g01 (geometry) ---

Geom Title=Geometry
Program Version=6.31

River Reach=LILAURELFK      ,Main
Reach XY= 30
2215413.95487995718075.599637738     2214961.929      718693.937
     2214051.928      719075.622     2213699.546      720274.077
     2212379.987      721482.661     2212107.931       721973.89
     2212260.628      721995.496     2212153.402      722336.231
     2212394.982      722662.5722212379.72110237723153.731954325
     2212704.354      723382.217     2212629.092      723559.152
     2212862.545      723591.288     2212800.962      723803.193
     2213039.566      723988.255     2212885.409      724076.279
     2213104.868      724440.022     2212948.966      724649.694
     2213118.061      724826.744     2213108.131      725298.285
     2213661.886      726151.654     2214056.878      726330.535
     2214078.598      727146.846      2214369.97      727486.322
     2214220.049      727698.942     2214468.239      727880.685
     2214397.528      728338.347     2214643.886      729110.045
     2214392.892      730071.069     2214167.166      730332.651

Type RM Length L Ch R = 1 ,17962   ,196.5,197.2,196.5
XS GIS Cut Line= 3
2215327.35061462717907.3399126782215467.46368263718207.026197014
 2215524.5467844718417.195799016
#Sta/Elev= 30
       0 1774.96    32.1 1766.74    46.2 1761.61    50.1 1760.76    68.2 1760.25
   147.7 1760.48  186.31 1759.26   190.8 1759.11   194.6 1759.27   200.3 1759.75
   218.4 1760.02   257.8 1759.61   271.4 1759.97   278.8 1759.72   284.6 1760.12
   297.9 1759.84   306.7 1760.38   346.2 1761.05   353.8 1761.88   366.2 1764.93
   370.4 1765.48   403.5 1766.57   428.4 1766.22   436.7 1766.53   457.4 1768.45
   482.3 1772.16   502.7 1771.36   511.3 1771.48     532 1776.57   548.6 1778.79
#Mann= 7 ,-1,0
       0      .1       0      80     .08       0     150      .1       0
  186.31    .045       0   194.6      .1       0     290     .06       0
  400.82      .1       0
Bank Sta=186.31,194.6
XS Rating Curve= 0 ,0
Exp/Cntr(USF)=0,0
Exp/Cntr=0.3,0.1

Type RM Length L Ch R = 1 ,17765   ,258,258.2,258
XS GIS Cut Line= 4
2215121.27534873718101.9314958612215197.99653567 718141.79250054
2215453.19290718 718251.135866572215515.46538185718417.195799016
#Sta/Elev= 30
       0  1776.2    21.3 1771.86    41.7  1770.7    75.8 1767.14    88.8 1763.72
    97.5 1759.87   101.9 1758.98   132.3 1758.18   145.4 1758.31   154.1    1759
   193.3 1759.17   210.7 1758.72   245.5 1759.34   250.41758.625   254.2 1758.29
   256.61758.598   267.7 1759.03   271.6 1759.72   280.3 1762.74   297.7 1764.21
   323.8 1764.36   345.6 1765.35   430.4 1765.89   451.7 1767.48   473.1 1769.86
     483 1772.19   510.9 1772.21   515.8 1773.04   528.6  1776.4   541.4 1778.29
#Mann= 7 ,-1,0
       0      .1       0   86.46     .08       0  156.46      .1       0
  196.46     .06       0   250.4    .045       0   256.6     .06       0
  384.09      .1       0
Bank Sta=250.4,256.6
XS Rating Curve= 0 ,0
Exp/Cntr(USF)=0,0
Exp/Cntr=0.3,0.1

Type RM Length L Ch R = 1 ,17507   ,184,184,184
XS GIS Cut Line= 2
2215067.88197018718209.6208834592215453.19290718718412.006426127
#Sta/Elev= 30
       0 1770.82    22.9 1766.66    33.5 1766.37    41.4 1764.81    53.2 1764.54
    59.1    1764    65.1 1762.87    73.9  1760.3    86.2 1759.44   117.8 1758.98
  121.811758.102   126.8 1757.68   130.2 1758.12   140.4 1759.55     151 1758.39
   168.7 1757.75   180.6 1758.15   217.2 1758.23   244.3 1758.91   275.9 1758.38
     285 1758.93   298.5 1761.08     308 1761.29   334.6 1763.25   352.8 1763.96
   361.8 1765.46   373.1 1765.43   384.4 1766.51     407 1769.58   435.2 1770.72
#Mann= 4 ,-1,0
       0     .05       0  121.81    .045       0   130.2     .06       0
     260      .1       0
Bank Sta=121.81,130.2
XS Rating Curve= 0 ,0
Exp/Cntr(USF)=0,0
Exp/Cntr=0.3,0.1

Type RM Length L Ch R = 1 ,17323   ,48.2,49.3,48.2
XS GIS Cut Line= 3
2215041.24232445 718340.856231792215124.46948684 718360.71725918
2215404.41539671718486.503765978
#Sta/Elev= 30
       0 1769.55       3 1769.14    15.4 1768.92    27.7 1767.44    35.9 1765.44
    44.1 1764.27    52.4 1763.99    60.6 1762.45    73.7 1758.98      77 1758.34
    85.6 1757.49    88.7  1757.6    94.8 1758.54   112.9 1758.42   124.7  1758.9
   140.2 1757.89  147.281757.894   190.5 1757.98   213.6 1758.42   233.1  1759.6
   256.3 1760.36   269.4 1762.23   276.3 1762.86   285.4 1763.52   308.9 1764.16
     322 1765.82   335.2 1766.92   373.1 1767.42   387.8 1766.98   392.5 1767.39
#Mann= 6 ,-1,0
       0     .05       0      60     .06       0   140.2    .045       0
  147.28     .06       0  165.56      .1       0  385.56     .06       0
Bank Sta=140.2,147.28
XS Rating Curve= 0 ,0
Exp/Cntr(USF)=0,0
Exp/Cntr=0.3,0.1

Type RM Length L Ch R = 1 ,17273   ,215.5,214.9,215.5
XS GIS Cut Line= 3
2215028.00163952718372.0664176882215111.22880192718391.927445077
2215391.17471178718517.713951875
#Sta/Elev= 30
       0 1770.02    16.6 1767.38    45.4 1764.85    56.5 1763.01      66 1760.87
    86.6 1757.46    95.4 1758.41   121.7 1758.05   150.8 1758.34  163.071757.728
   169.9 1757.72   187.1 1758.24   196.2 1758.87   209.4 1758.32   213.8 1758.78
   218.2 1760.23   222.5  1760.3   229.4 1759.67   248.9 1760.46   264.3 1762.08
   283.9 1763.12   289.9 1764.44   301.5 1769.78   305.9 1770.81   310.2 1771.06
   345.3 1768.37   371.6 1767.66   384.8 1768.02   389.2 1767.84   392.5 1767.27
#Mann= 5 ,-1,0
       0     .06       0  163.07    .045       0   169.9     .06       0
  185.56      .1       0  392.47     .06       0
Bank Sta=163.07,169.9
XS Rating Curve= 0 ,0
Exp/Cntr(USF)=0,0
Exp/Cntr=0.3,0.1

Type RM Length L Ch R = 1 ,17058   ,328.6,328.6,328.6
XS GIS Cut Line= 2
2215011.92366497718428.8122102282215178.37798976718724.836094648
#Sta/Elev= 30
       0  1769.6       5 1768.38     9.3 1767.09    12.2 1765.95    18.8 1762.52
    23.4 1759.71      25 1759.07      28  1758.3    32.5 1758.06    56.3 1758.18
    64.7 1757.78    73.8 1757.66    78.4 1757.01    82.7 1756.77   84.771757.007
    92.2 1757.94   133.5 1757.62   138.5 1757.81   147.3 1759.06   151.9 1759.36
   197.7 1759.84   250.1 1761.45   257.4  1761.4   266.6 1761.71   289.5 1761.07
   298.7 1761.33   303.3  1762.3   312.5 1765.03   323.6  1768.8   339.6 1774.96
#Mann= 6 ,-1,0
       0     .06       0      50     .05       0    78.4    .045       0
   84.77     .05       0     160      .1       0     270     .08       0
Bank Sta=78.4,84.77
XS Rating Curve= 0 ,0
Exp/Cntr(USF)=0,0
Exp/Cntr=0.3,0.1

Type RM Length L Ch R = 1 ,16730   ,171.6,171.6,171.6
XS GIS Cut Line= 2
2214869.11342041718594.320771805 2215025.1643499718764.558149426
#Sta/Elev= 30
       0 1768.35     3.9 1766.97    14.7 1762.39    18.3 1761.17    25.6 1759.22
      31  1758.2      40 1757.51    47.3 1757.56    57.8 1757.25    66.5 1757.59
    81.5 1757.17    87.4 1757.33   114.6 1757.17   128.7  1757.4  133.621756.373
   134.4  1756.2   137.3 1756.08   140.1 1756.37   142.9 1756.91   146.6 1757.23
   158.4  1756.7   177.5 1757.12   182.9 1757.34   193.9 1758.41   199.2 1759.52
   205.2  1761.4   215.5 1766.28   223.6 1769.43   226.4 1770.67   230.9 1773.09
#Mann= 7 ,-1,0
       0     .05       0      50      .1       0     100     .08       0
  133.62    .045       0   140.1     .08       0     190     .07       0
     230     .08       0
Bank Sta=133.62,140.1
XS Rating Curve= 0 ,0
Exp/Cntr(USF)=0,0
Exp/Cntr=0.3,0.1

Type RM Length L Ch R = 1 ,16558   ,130.8,131.2,130.8
XS GIS Cut Line= 2
2214792.34780567718655.6832899362214867.25225183718814.855238012
#Sta/Elev= 30
       0  1766.5     1.7 1766.53     6.1 1766.21      10    1765    14.9  1762.6
    19.3 1759.85      22 1758.48    23.8 1757.73    28.2 1757.02    32.6 1756.87
    37.1 1756.96    43.1 1755.97    45.9 1755.64   47.99 1755.97    52.1 1756.75
    55.1 1757.08    70.1 1756.94    81.2 1756.65    90.1 1756.71    98.9 1756.21
   112.2 1756.75   129.9 1756.93   138.7 1756.86   143.1 1757.61   148.3 1759.24
     152 1760.57   165.2 1766.26   169.6  1768.3   174.1 1770.61   175.9 1771.68
#Mann= 5 ,-1,0
       0     .05       0      10     .07       0    43.1    .045       0
   47.99     .07       0     120     .08       0
Bank Sta=43.1,47.99
XS Rating Curve= 0 ,0
Exp/Cntr(USF)=0,0
Exp/Cntr=0.3,0.1

Type RM Length L Ch R = 1 ,16427   ,229.8,229.3,229.8
XS GIS Cut Line= 3
2214646.05461432718690.086710502 2214662.8891969718742.643096547
2214826.87526548718839.068696062
#Sta/Elev= 30
       0 1777.46    10.5 1771.62    16.9 1768.73      20 1766.97    24.2 1763.46
    28.4 1761.11    36.8 1758.92    45.2 1758.36    60.2 1757.92    70.6  1756.4
    81.4  1756.8    90.1 1756.12   103.1 1756.35   112.4 1755.52   117.61753.853
   121.6 1753.17   124.61753.827   130.9 1755.02   135.6 1755.48   151.5 1755.28
   170.7 1755.93     182 1755.97   189.5 1756.31   195.3 1756.89   201.2 1758.16
   219.1 1764.07   227.5 1767.46   239.1 1772.98   241.7 1773.78   245.4 1774.02
#Mann= 5 ,-1,0
       0     .05       0   95.19     .07       0  105.19     .08       0
   117.6    .045       0   124.6     .08       0
Bank Sta=117.6,124.6
XS Rating Curve= 0 ,0
Exp/Cntr(USF)=0,0
Exp/Cntr=0.3,0.1

Type RM Length L Ch R = 1 ,16198   ,176,176,176
XS GIS Cut Line= 2
2214533.73986485718758.0105091832214625.48163884718931.296157288
#Sta/Elev= 30
       0 1767.19     3.6 1766.72     8.1 1766.66    12.6 1766.47    17.2 1765.65
    26.2 1762.03    30.8 1760.34    33.7 1758.56    35.3 1757.47    39.8 1754.11
    42.6  1753.1    44.3  1752.7    45.6 1752.71   49.041753.105    53.4 1754.18
    57.9  1754.9    63.3 1755.02    82.1 1755.81    98.6 1756.34   103.2 1756.45
   117.2 1756.36   130.3 1756.99   152.9 1757.58   157.5  1758.5   166.9 1761.26
   169.9 1762.27   180.1 1766.26   189.2 1770.01   193.5 1771.45   196.1 1771.79
#Mann= 4 ,-1,0
       0     .05       0    42.6    .045       0   49.04     .05       0
     120     .08       0
Bank Sta=42.6,49.04
XS Rating Curve= 0 ,0
Exp/Cntr(USF)=0,0
Exp/Cntr=0.3,0.1

Type RM Length L Ch R = 1 ,16022   ,140.8,180.4,140.8
XS GIS Cut Line= 2
2214453.64573224 718793.143843822214490.24676843  719009.3453134
#Sta/Elev= 30
       0 1769.06     8.1 1768.99    12.2 1768.67    16.3 1767.54    24.4 1763.72
    28.4 1761.08    32.5 1758.02    36.5 1756.09    40.6  1755.3    44.7 1755.04
    52.8 1755.03    77.1 1755.45    85.2 1755.38    95.9 1754.96   106.3 1755.15
   116.7 1754.68   133.9 1754.84     142 1754.42   146.1 1753.88   151.4 1752.75
   154.2 1752.44   158.9 1752.75   166.4 1754.64   174.5 1755.31   186.1 1755.84
   190.7 1756.83   198.8 1760.24     211 1765.78   215.1 1767.86   219.3  1769.6
#Mann= 4 ,-1,0
       0     .05       0      70     .07       0   151.4    .045       0
   158.9     .07       0
Bank Sta=151.4,158.9
XS Rating Curve= 0 ,0
Exp/Cntr(USF)=0,0
Exp/Cntr=0.3,0.1

Type RM Length L Ch R = 1 ,15841   ,132.6,261.2,132.6
XS GIS Cut Line= 3
2214293.44031793718838.6399529462214360.67942074719059.395782246
2214388.65710347719097.231209379
#Sta/Elev= 30
       0 1767.22     6.8 1765.02      11 1764.67    23.6 1764.53    31.9 1763.01
    36.3 1763.06    40.3  1762.7    44.5 1761.35    52.3 1757.97    55.5 1757.12
    65.4  1756.5    69.6 1755.88    73.7 1753.29    75.41752.643    77.9 1751.94
    83.81752.562    90.8 1754.19   115.6  1754.2   123.9 1754.79   132.3 1754.99
   144.8 1753.95   165.7 1754.92   178.3 1755.02   186.6 1755.43   222.2 1755.81
   225.4 1756.28   230.8 1757.89   263.1 1769.05   267.8 1769.51   277.8  1769.3
#Mann= 6 ,-1,0
       0     .05       0      30      .1       0    75.4    .045       0
    83.8      .1       0     130     .07       0     230     .08       0
Bank Sta=75.4,83.8
XS Rating Curve= 0 ,0
Exp/Cntr(USF)=0,0
Exp/Cntr=0.3,0.1

Type RM Length L Ch R = 1 ,15580   ,299.1,251.8,299.1
XS GIS Cut Line= 3
2214055.75264173718793.219868133  2214098.314682718980.373324746
2214304.21188767719185.247188768
#Sta/Elev= 30
       0 1766.87    20.6 1763.13    36.9 1761.74    45.1 1762.43    49.2 1762.14
    53.3  1760.8    61.5 1756.82    65.6 1756.68    70.5 1757.48    77.9 1757.75
    98.4 1756.05   102.5 1755.91   110.9 1756.77   127.1 1755.51   184.6  1756.2
   194.6 1755.83   211.5  1754.2   292.8 1753.75     3001752.267   301.8 1751.83
     307 1752.15   313.1 1753.71   318.7 1754.39   374.5 1754.34   391.6 1753.68
   414.2 1754.36   425.6 1756.64   454.1 1768.39   465.4 1768.69   482.4 1767.71
#Mann= 5 ,-1,0
       0      .1       0     300    .045       0     307      .1       0
  351.93     .07       0  441.93     .08       0
Bank Sta=300,307
XS Rating Curve= 0 ,0
Exp/Cntr(USF)=0,0
Exp/Cntr=0.3,0.1

Type RM Length L Ch R = 1 ,15328   ,318.5,320.2,318.5
XS GIS Cut Line= 4
2213773.69449092719062.4539186562213874.42906797719128.122353429
2214148.71183071719172.5360708442214266.62446591719222.919396141
#Sta/Elev= 30
       0 1762.97     7.7  1762.7    22.1 1760.98    45.9 1756.08    52.9 1756.61
    61.6 1755.89     122 1755.74   134.2 1755.04   146.3 1753.57   174.7 1753.01
   231.4 1753.74     280 1753.57   292.2 1752.77   320.6 1752.12   326.11751.027
   328.7  1750.5   332.7 1751.05   336.8 1752.42   340.8 1752.88     357 1753.64
   372.5 1753.72   401.9 1754.92   419.3 1753.57     428 1753.62     453  1755.1
   474.4 1762.45   484.5 1766.75   489.6 1768.28   501.9 1768.47   526.3 1767.28
#Mann= 7 ,-1,0
       0     .05       0      60     .07       0  170.25      .1       0
   326.1    .045       0   332.7      .1       0  360.25     .07       0
   468.1     .08       0
#XS Ineff= 2 , 0
          231.63 1756.09
Permanent Ineff=
       F       F
Bank Sta=326.1,332.7
XS Rating Curve= 0 ,0
Exp/Cntr(USF)=0,0
Exp/Cntr=0.3,0.1

Type RM Length L Ch R = 1 ,15008   ,189.9,189.9,189.9
XS GIS Cut Line= 2
 2213731.0727375719270.2158236882214017.92973887719446.077904925
#Sta/Elev= 30
       0 1765.32    10.7 1764.68    24.8 1762.75    43.5 1759.38    55.3 1758.45
    57.6 1758.07    66.9 1755.36    76.4 1754.21    95.1 1753.54   113.9 1753.75
   132.7 1753.02   142.6 1753.14   151.4 1753.68     160 1752.71     189 1751.54
     220 1752.55   241.5 1752.08   250.2 1750.95   253.1  1750.8   264.7 1751.29
   281.2 1751.47   282.8 1751.39  290.081749.926   293.8 1749.61   296.9 1749.93
   306.3 1753.47   315.6 1758.63   329.7 1765.56   334.4 1766.64   336.5 1766.67
#Mann= 6 ,-1,0
       0     .08       0     100      .1       0     220     .07       0
  290.08    .045       0   296.9     .07       0  336.47     .08       0
#XS Ineff= 2 , 0
          104.67  1755.6
Permanent Ineff=
       F       F
Bank Sta=290.08,296.9
XS Rating Curve= 0 ,0
Exp/Cntr(USF)=0,0
Exp/Cntr=0.3,0.1

Type RM Length L Ch R = 1 ,14818   ,395.6,395.6,395.6
XS GIS Cut Line= 4
2213600.60635418719808.7527084512213697.49679449719790.956505128
2213944.86382294 719458.28772623 2214000.6495815 719486.82927712
#Sta/Elev= 30
       0 1792.48      24  1787.1    48.4 1777.11    76.8 1763.47    80.9 1761.99
    93.1 1763.05   133.1 1762.77   147.4 1760.74   163.3 1759.87   190.1  1756.8
   243.8 1753.53   261.8 1754.03   336.1 1753.68     350 1753.16   381.9 1753.57
   384.9 1753.31   389.8 1750.47  394.411748.817     398 1748.14   410.5 1748.81
   434.7 1752.11   451.6 1753.36   461.9 1753.31   484.8 1751.79   514.7 1752.07
   535.5 1754.77   539.3 1756.13   557.2 1765.05   559.3 1765.58   575.7 1766.06
#Mann= 9 ,-1,0
       0     .05       0      20      .1       0  138.51     .08       0
  158.51     .07       0  288.51     .06       0  298.51     .07       0
  394.41    .045       0   410.5      .1       0  468.51     .07       0
#XS Ineff= 2 , 0
          378.72 1758.11   462.4         1757.04
Permanent Ineff=
       F       F
Bank Sta=394.41,410.5
XS Rating Curve= 0 ,0
Exp/Cntr(USF)=0,0
Exp/Cntr=0.3,0.1

Type RM Length L Ch R = 1 ,14423   ,319.9,319.9,319.9
XS GIS Cut Line= 4
2213544.15481988719958.9253769842213744.83271797720057.890063663
2214010.36255154719723.9239415432214059.66159398719758.952208543
#Sta/Elev= 30
       0 1783.95     7.7 1778.43    22.6  1764.1    26.8 1762.67    44.6 1761.36
      58 1756.74    91.3  1760.9   124.9 1762.02   142.7  1759.8   160.6  1761.9
     195 1762.48   201.8  1761.5   223.8 1753.93   248.4 1753.23   297.8  1755.2
   303.5 1754.56   312.7 1751.79   329.1 1754.21   351.9 1752.83  376.031748.805
   383.1 1748.08  385.49 1748.86   393.3 1753.94   396.2 1754.22   434.8 1752.83
   550.5 1754.41   576.2 1755.18   650.4 1759.98   669.8 1767.48   710.9  1779.1
#Mann= 7 ,-1,0
       0     .07       0      90     .08       0  343.75     .07       0
  373.75     .08       0  376.03    .045       0  385.49     .08       0
  690.41     .07       0
#XS Ineff= 2 , 0
          327.25 1756.83  399.93         1756.71
Permanent Ineff=
       F       F
Bank Sta=376.03,385.49
XS Rating Curve= 0 ,0
Exp/Cntr(USF)=0,0
Exp/Cntr=0.3,0.1

Type RM Length L Ch R = 1 ,14103   ,353.6,376.4,353.6
XS GIS Cut Line= 3
2213495.47781213720033.4844703722213743.01089893720237.816027874
2213841.09004653720249.492116875
#Sta/Elev= 30
       0 1789.67     6.1 1786.05    21.7 1771.57    26.8 1767.07    28.7 1765.86
      32 1764.37    47.6 1762.55    62.8 1757.44    68.5 1757.88    79.8 1760.07
    89.1 1760.61   116.8 1761.35   120.2 1761.14     131 1759.22   135.8    1759
   151.3 1761.27   173.6 1761.94     188 1761.71   193.5 1761.26   213.4 1757.91
   234.3 1752.67   250.3 1749.61   270.6 1748.08   275.8 1747.82  277.871748.079
   312.1 1752.68   322.1 1752.82   362.4  1763.5   382.6 1767.06   419.7 1777.67
#Mann= 7 ,-1,0
       0      .1       0      10     .07       0      40     .08       0
     170     .07       0   270.6    .045       0  277.87     .07       0
     290      .1       0
Bank Sta=270.6,277.87
XS Rating Curve= 0 ,0
Exp/Cntr(USF)=0,0
Exp/Cntr=0.3,0.1

Type RM Length L Ch R = 1 ,13726   ,274.5,262.1,274.5
XS GIS Cut Line= 3
2213391.60799479720351.6307847332213701.97190037720636.886060476
2213835.64224386720732.247385093
#Sta/Elev= 30
       0 1759.91     4.3 1759.48    12.8 1757.66    18.5 1757.14    31.8 1759.52
    38.3 1760.03    60.5 1760.53    75.1 1760.24    87.7 1757.39   114.7  1748.9
   129.3  1747.4   134.6 1747.08     1381747.345   144.2 1748.48   150.1 1748.83
   174.2 1748.68   191.4 1749.09   219.5 1748.22   253.5 1748.73   273.3 1748.57
   321.4 1750.31     344  1751.9   369.5 1755.19   391.9 1757.42   429.2 1759.38
   453.7 1760.05   504.7 1763.36   540.9 1764.77   561.8  1766.1   585.7 1768.94
#Mann= 3 ,-1,0
       0     .08       0   129.3    .045       0     138      .1       0
Bank Sta=129.3,138
XS Rating Curve= 0 ,0
Exp/Cntr(USF)=0,0
Exp/Cntr=0.3,0.1

Type RM Length L Ch R = 1 ,13464   ,350.7,340.4,350.7
XS GIS Cut Line= 3
2213246.76250633  720531.36488762213392.28151403720719.212361568
2213413.33496943720835.679964421
#Sta/Elev= 30
       0 1758.03     5.2 1757.03     8.8  1756.8    12.4 1757.21    22.3 1759.18
    27.6 1759.69    50.8 1760.31      65 1759.98    67.9 1759.62    78.2 1757.22
   119.2 1746.78   124.9 1746.23   130.11746.633   147.7 1747.46   159.1 1746.78
   170.5 1746.52   179.4  1747.1   190.5 1746.79   201.9 1747.27   207.6 1748.37
   214.8 1750.78   221.8 1752.43     230  1753.8   247.7 1756.25   259.9 1757.62
   272.1 1759.55   288.4 1763.17   332.2    1772   349.4 1775.81     356 1776.64
#Mann= 3 ,-1,0
       0     .08       0   119.2    .045       0   130.1      .1       0
Bank Sta=119.2,130.1
XS Rating Curve= 0 ,0
Exp/Cntr(USF)=0,0
Exp/Cntr=0.3,0.1

Type RM Length L Ch R = 1 ,13124   ,252.5,252.5,252.5
XS GIS Cut Line= 2
2213043.80817588720772.759017223 2213189.5590811720961.754696512
#Sta/Elev= 30
       0  1760.4     6.3 1760.88    26.2 1761.44    39.9 1761.35    43.3 1761.04
      46  1760.6    51.9 1759.19    63.3 1755.91    72.7 1752.71    77.6 1750.75
    86.1    1747   88.48  1746.3    91.8 1745.63    96.5 1745.94    98.71746.281
   103.2  1747.4   108.9  1749.3   114.6 1750.83   126.8 1752.94   136.9 1755.71
     142 1756.68     147 1758.21   152.1 1760.09   167.2 1766.41   172.3 1768.09
   177.3 1769.49   192.5 1772.76   207.6 1776.35   216.8 1778.18   238.7 1783.09
#Mann= 4 ,-1,0
       0     .08       0      70      .1       0   88.48    .045       0
    98.7      .1       0
Bank Sta=88.48,98.7
XS Rating Curve= 0 ,0
Exp/Cntr(USF)=0,0
Exp/Cntr=0.3,0.1

Type RM Length L Ch R = 1 ,12871   ,261,261,261
XS GIS Cut Line= 2
2212882.26820567720943.850348908 2212992.7826283721097.609545618
#Sta/Elev= 30
       0 1762.58    13.8 1762.94    23.8 1762.94    28.1 1762.78      31 1762.37
    42.4  1758.3      46 1756.85    50.9 1754.02    60.7 1746.99    64.9 1744.75
    65.7 1744.44    67.5 1744.14    70.6  1743.8      74 1744.13    76.8 1744.89
    80.5 1746.57    85.4 1748.43    90.3 1749.06   102.6 1750.18   108.4 1750.84
     110 1751.13   119.9 1753.95   122.7    1755   144.5 1765.71   151.4 1768.67
   162.8 1774.03   171.4 1778.41   174.3 1779.68   182.9 1782.67   189.4 1785.25
#Mann= 5 ,-1,0
       0     .08       0    67.5    .045       0      74     .08       0
      90     .07       0     100     .06       0
Bank Sta=67.5,74
XS Rating Curve= 0 ,0
Exp/Cntr(USF)=0,0
Exp/Cntr=0.3,0.1

Type RM Length L Ch R = 1 ,12610   ,271,271,271
XS GIS Cut Line= 2
2212704.48413447721104.0161788142212794.17699922721246.563767431
#Sta/Elev= 30
       0 1764.04    10.8 1764.27    20.3 1764.15      22 1764.05      25 1763.68
    29.5 1762.46    34.5 1760.35    48.6  1753.8      52 1752.08    58.6 1748.54
    67.3 1743.51    70.2  1742.7    73.1  1742.3    74.5 1742.34   76.531742.698
    78.9 1743.68    81.7 1745.17    84.7 1747.04    90.5 1750.85    93.4 1752.26
    96.3 1753.45     105 1755.77   110.8 1757.46   113.7  1758.1   119.5 1759.16
   124.2 1759.79   134.1 1760.55   138.4 1761.17   149.6 1763.15   168.4 1765.49
#Mann= 4 ,-1,0
       0     .08       0    70.2    .045       0   76.53     .08       0
     140     .06       0
Bank Sta=70.2,76.53
XS Rating Curve= 0 ,0
Exp/Cntr(USF)=0,0
Exp/Cntr=0.3,0.1

Type RM Length L Ch R = 1 ,12339   ,344.9,344.9,344.9
XS GIS Cut Line= 2
2212499.27180392721247.9824999642212649.82768403721464.206370337
#Sta/Elev= 30
       0 1765.12    22.6 1765.69    33.1 1765.69    38.9  1765.4    43.6 1764.62
    50.2 1762.53    73.3 1752.57    84.8 1748.33    94.1 1746.27   108.7  1745.2
   113.6 1744.19   118.4 1742.04   120.6 1741.45   123.3  1740.9   128.2 1740.91
  131.881741.443   133.1 1741.62   137.9  1743.7   142.8 1744.97   173.9 1748.26
   186.7 1749.04   190.6 1749.78   197.6 1752.55   205.5 1756.09   214.1 1759.09
   220.8 1761.03   235.4 1763.73     240 1765.09   254.4 1771.22   263.5 1775.38
#Mann= 6 ,-1,0
       0     .08       0      90     .07       0   120.6    .045       0
  131.88     .07       0     210      .1       0     240     .07       0
Bank Sta=120.6,131.88
XS Rating Curve= 0 ,0
Exp/Cntr(USF)=0,0
Exp/Cntr=0.3,0.1

Type RM Length L Ch R = 1 ,11994   ,150.9,150.9,150.9
XS GIS Cut Line= 2
2212220.58325988721469.0113452342212515.28838691721738.089939476
#Sta/Elev= 30
       0 1767.72      18 1767.54      24 1766.45    37.4  1761.1    56.5 1752.48
    59.6 1751.06    71.4 1744.63    73.4 1743.99    77.4 1743.11    89.2 1742.87
    98.9 1740.75   107.8 1740.27   124.8 1739.85   200.9 1739.92   205.3 1740.28
   207.9 1740.97   216.1 1744.26   219.7 1745.37   231.6  1747.5   237.5 1749.41
   243.3 1750.81   255.3 1752.64   264.9 1753.38   281.1 1755.29   322.6 1761.95
   351.5 1767.39   356.6 1768.75   379.9 1776.91   389.4 1781.77   399.1 1788.04
#Mann= 5 ,-1,0
       0     .08       0      30     .07       0      70      .1       0
   107.8    .045       0   205.3      .1       0
Bank Sta=107.8,205.3
XS Rating Curve= 0 ,0
Exp/Cntr(USF)=0,0
Exp/Cntr=0.3,0.1

Type RM Length L Ch R = 1 ,11843   ,42.9,42.9,42.9
XS GIS Cut Line= 3
2212059.97120797721612.8589998912212224.95434555721702.181080742
2212483.46295601721752.621785223
#Sta/Elev= 30
       0 1766.68    32.8 1765.79    42.7 1764.81   104.8 1755.43   127.3 1751.19
   141.2 1747.88   154.9  1745.9   168.6 1744.53   186.7 1743.83   211.3 1744.87
   223.5 1744.58   239.8  1743.5     252  1743.5   258.8 1740.76   260.2 1740.09
   264.3 1739.94  265.991740.781   272.4  1743.6   280.6 1743.72   292.8 1742.78
   304.4 1743.86   321.3 1746.85   328.6 1747.71   337.6  1746.6   341.7  1746.8
     358 1750.07   382.4 1755.66   427.3 1763.67   439.5 1768.32     451 1774.18
#Mann= 4 ,-1,0
       0     .08       0      10      .1       0   258.8    .045       0
  265.99      .1       0
#XS Ineff= 2 , 0
          211.72 1746.36
Permanent Ineff=
       F       F
Bank Sta=258.8,265.99
XS Rating Curve= 0 ,0
Exp/Cntr(USF)=0,0
Exp/Cntr=0.3,0.1

Type RM Length L Ch R = 1 ,11801   ,132.3,132.3,132.3
XS GIS Cut Line= 3
2212046.83560785721653.3166482772212211.81874542721742.638729128
2212470.32735588721793.079433609
#Sta/Elev= 30
       0  1771.4    18.6 1767.58    28.8 1764.96    65.2 1759.27   101.6 1752.12
   119.8 1747.75   134.1 1742.91     138 1742.31   151.6 1741.04   169.1 1741.82
     188 1741.46   196.1 1742.04   224.7 1742.36     245 1743.51   249.1 1743.36
   251.5 1742.76   257.3 1740.36   260.8 1739.49   265.1 1739.16   270.9 1739.52
   273.6 1739.98   281.7 1743.42     289 1743.46   299.2 1742.84   326.5 1747.91
   355.1 1754.84   379.5 1757.76   394.7 1760.24     422 1767.02     451 1775.91
#Mann= 3 ,-1,0
       0      .1       0   260.8    .045       0   270.9      .1       0
#XS Ineff= 2 , 0
          245.15 1747.25
Permanent Ineff=
       F       F
Bank Sta=260.8,270.9
XS Rating Curve= 0 ,0
Exp/Cntr(USF)=0,0
Exp/Cntr=0.3,0.1

Type RM Length L Ch R = 1 ,11668   ,182.9,182.9,182.9
XS GIS Cut Line= 2
2212049.46272787721789.4014655732212332.14084257721919.706618815
#Sta/Elev= 30
       0 1761.12    33.8 1753.57    42.6 1751.05    55.8 1748.59    73.5 1746.38
    89.3 1744.01   104.3 1742.81   123.7 1742.49   135.1 1741.32   152.7 1741.01
   164.7 1741.32   167.7  1740.9   174.8 1738.83  178.211738.213   183.6 1737.91
  191.561738.208   196.8 1740.34   200.1 1740.83   214.4 1740.11   218.8 1740.13
   227.6 1741.26     232  1741.5   240.8 1741.22   246.1 1741.49   249.6 1742.36
   264.2 1749.07   267.2 1750.33   273.2 1752.29   302.5 1758.59   311.3 1759.92
#Mann= 3 ,-1,0
       0      .1       0  178.21    .045       0  191.56      .1       0
Bank Sta=178.21,191.56
XS Rating Curve= 0 ,0
Exp/Cntr(USF)=0,0
Exp/Cntr=0.3,0.1

Type RM Length L Ch R = 1 ,11485   ,338.5,338.4,338.5
XS GIS Cut Line= 2
2211990.66843038721995.4065958322212333.98047526721947.172672173
#Sta/Elev= 30
       0 1758.55     9.6 1756.85    41.9  1753.2    58.1 1750.92    62.1 1750.05
    67.1 1748.47    81.2 1741.31    84.8 1740.25    90.4 1739.58   102.5 1739.94
     106 1739.69   111.9 1738.02   114.6 1737.52  123.081738.005   130.8  1740.5
   134.8 1740.83   162.7 1739.88   175.2 1741.43   183.3 1741.84   187.3  1741.9
   199.4  1741.1   223.7 1740.57     252 1740.45     260 1741.92     276  1747.4
   288.3 1750.67   304.5 1753.78   328.7    1759   336.8 1759.97   346.7 1763.26
#Mann= 3 ,-1,0
       0      .1       0   111.9    .045       0  123.08      .1       0
Bank Sta=111.9,123.08
XS Rating Curve= 0 ,0
Exp/Cntr(USF)=0,0
Exp/Cntr=0.3,0.1

Type RM Length L Ch R = 1 ,11147   ,230.6,230.8,230.6
XS GIS Cut Line= 3
2211973.40212836722064.7989095612212086.29196411722059.677091914
 2212307.4991054722155.240578156
#Sta/Elev= 30
       0 1763.86     6.8 1761.77    22.8 1757.87    50.8 1753.27    58.8 1752.22
    70.8 1749.67    86.9 1747.43     104 1745.54   124.7 1743.47   133.8 1743.14
   141.2 1742.09   149.9 1740.02   154.3 1739.61   164.3 1739.45   193.5 1740.54
   209.9 1740.68   219.6 1740.31   237.1 1740.35   243.4  1739.9   245.8 1739.37
   250.1 1737.75     2521737.403   258.6 1736.85   261.6 1737.45   273.8 1741.32
   282.9 1745.35   289.3 1747.41   298.3 1748.95   328.6 1752.53     354 1756.91
#Mann= 3 ,-1,0
       0      .1       0     252    .045       0   261.6      .1       0
Bank Sta=252,261.6
XS Rating Curve= 0 ,0
Exp/Cntr(USF)=0,0
Exp/Cntr=0.3,0.1

Type RM Length L Ch R = 1 ,10916   ,229.1,237.9,229.1
XS GIS Cut Line= 2
 2211982.1565615722210.0948442782212345.32963376722289.538953835
#Sta/Elev= 30
       0 1761.74     6.2 1760.24    38.9  1756.2    55.3 1754.58    71.7 1751.95
    88.1 1748.58   100.3 1745.01   108.5 1742.12   112.6 1741.08   116.7 1740.63
   153.6 1739.44   169.9 1739.42   178.1 1739.09   198.6 1739.81     215 1739.42
   243.6 1739.93   280.5 1739.77   284.6 1739.29  291.131737.101   292.8 1736.54
   296.9  1736.4  301.691737.093   305.1 1738.53   309.2 1740.76   313.4 1743.52
   316.7 1744.99   325.5 1747.37   341.9 1750.56   366.5 1752.81   371.8 1753.53
#Mann= 4 ,-1,0
       0      .1       0  291.13    .045       0  301.69      .1       0
     370     .06       0
Bank Sta=291.13,301.69
XS Rating Curve= 0 ,0
Exp/Cntr(USF)=0,0
Exp/Cntr=0.3,0.1

Type RM Length L Ch R = 1 ,10678   ,132.7,122.9,132.7
XS GIS Cut Line= 3
2212010.89533191722402.1821348222212288.79469721722352.706630349
2212386.04807149 722288.21837907
#Sta/Elev= 30
       0 1758.41    21.6 1757.55    25.7 1756.88    33.8 1754.27    39.9 1753.06
   105.4 1745.09   123.2 1744.09   139.4 1739.69  144.73 1737.26   147.6 1736.25
   151.6 1736.18   155.7 1736.37   159.8 1737.29   163.8 1738.46   171.9    1739
   188.2 1738.88   216.6 1739.72     233 1741.32   245.1 1744.17   250.3 1743.71
   273.5  1743.7   281.6 1744.88   291.1 1747.79   298.8 1746.66   317.6  1745.9
   332.1  1749.5   353.5 1751.95   367.9 1754.61   388.3 1757.25     399 1759.76
#Mann= 5 ,-1,0
       0     .06       0      10      .1       0  144.73    .045       0
   159.8      .1       0     240     .06       0
Bank Sta=144.73,159.8
XS Rating Curve= 0 ,0
Exp/Cntr(USF)=0,0
Exp/Cntr=0.3,0.1

Type RM Length L Ch R = 1 ,10555   ,37.3,37.3,37.3
XS GIS Cut Line= 4
2212024.40765716722482.6941589472212149.53212971722492.908401604
2212269.54948094722427.3670112192212392.97157971722312.456781324
#Sta/Elev= 30
       0 1761.59    15.8 1759.37    23.8 1759.37    43.9 1755.66      68  1753.5
   104.1 1748.88   112.1 1747.28   125.5  1743.3     145 1742.84   160.5 1741.79
   203.9 1742.96   208.4 1742.04  214.751737.619   216.8 1736.75   219.7  1736.6
  222.521737.636   224.3 1738.23   228.8 1740.88   233.5 1742.02   237.9 1742.32
   250.2 1741.92   268.5  1744.2   271.3 1743.71   298.7  1744.1   347.7 1747.21
   371.2 1749.59   388.8 1752.71   400.5 1753.32     410 1755.25   430.9 1757.58
#Mann= 5 ,-1,0
       0     .06       0  214.75    .045       0  222.52     .06       0
  235.54      .1       0  302.29     .06       0
Bank Sta=214.75,222.52
XS Rating Curve= 0 ,0
Exp/Cntr(USF)=0,0
Exp/Cntr=0.3,0.1

Type RM Length L Ch R = 1 ,10518   ,124.2,124.2,124.2
XS GIS Cut Line= 4
2212030.79155882722518.4440082472212155.91603137722528.658250905
 2212275.9333826 722463.116860522212399.35548137722348.206630625
#Sta/Elev= 30
       0 1761.49    21.5 1760.31    57.6 1756.11    81.6 1751.44      99 1746.69
   125.5  1744.8   132.8 1742.74   144.1 1741.87   198.8 1740.86   203.3    1739
  207.431736.425   212.4 1735.43     217 1735.58   219.7 1736.52   228.5 1740.22
   234.4 1741.84   248.9 1744.24   294.5 1745.61   300.9  1747.4   306.2 1747.85
   314.8 1747.65   337.4 1748.85   353.2 1750.46   362.9 1752.27   371.4  1752.5
   382.5 1754.41   388.3 1754.78   399.2 1752.29     406 1751.69   430.9 1753.86
#Mann= 6 ,-1,0
       0      .1       0  185.54     .06       0  207.43    .045       0
   219.7     .06       0  225.54      .1       0  362.29     .06       0
Bank Sta=207.43,219.7
XS Rating Curve= 0 ,0
Exp/Cntr(USF)=0,0
Exp/Cntr=0.3,0.1

Type RM Length L Ch R = 1 ,10394   ,239.5,239.5,239.5
XS GIS Cut Line= 2
2212137.61551328722665.6993398912212441.48923233722506.527391814
#Sta/Elev= 30
       0 1759.75      21 1757.09    25.5 1756.17    34.5 1752.83      39 1751.91
    52.6 1750.86    70.6 1750.53    88.7 1748.57    94.1 1747.24   104.6  1743.1
   113.2 1738.87   120.3 1734.88  121.141734.696   124.8 1734.28   130.4 1734.69
   138.6 1736.02   151.9  1736.7   156.3 1737.66   160.9 1739.18   165.4 1739.65
   190.8 1738.71   210.6 1738.48   242.2  1736.4   246.7 1737.59   259.7 1745.39
   264.8 1747.78   269.3 1749.28   287.4 1752.38   323.5 1756.28     343 1757.79
#Mann= 3 ,-1,0
       0      .1       0  121.14    .045       0   130.4      .1       0
#XS Ineff= 2 , 0
                          167.07         1743.18
Permanent Ineff=
       F       F
Bank Sta=121.14,130.4
XS Rating Curve= 0 ,0
Exp/Cntr(USF)=0,0
Exp/Cntr=0.3,0.1

Type RM Length L Ch R = 1 ,10154   ,338.9,339.1,338.9
XS GIS Cut Line= 2
2212184.67032493722754.0313460552212504.12811997722714.099121674
#Sta/Elev= 30
       0 1760.14    11.1 1757.82    19.7 1756.52    27.7 1755.76    36.2 1755.55
    68.4 1749.67    92.2  1746.5   120.4 1744.36   140.6 1742.28   156.7 1741.08
   184.9  1739.7   201.1 1738.22   209.1 1737.85   213.2 1737.06   221.2 1734.15
   222.5 1733.91   225.2 1733.45   229.3 1733.25   233.3  1733.5  234.451733.914
   237.3 1734.96   241.4 1737.51   249.4 1744.03   256.4 1747.35   261.5 1749.12
   273.6 1752.45   297.7 1757.77   305.9 1758.85   309.9 1759.69   321.9 1760.56
#Mann= 3 ,-1,0
       0      .1       0   222.5    .045       0  234.45      .1       0
Bank Sta=222.5,234.45
XS Rating Curve= 0 ,0
Exp/Cntr(USF)=0,0
Exp/Cntr=0.3,0.1

Type RM Length L Ch R = 1 ,9815    ,171.9,172.4,171.9
XS GIS Cut Line= 3
2212280.08991892722986.2298359712212441.92051247722984.128139951
2212551.20870551  722936.8399795
#Sta/Elev= 30
       0 1751.28    24.1 1750.21    28.1 1748.94    31.4 1746.86    36.1 1744.36
    40.1 1742.84    64.1 1735.36    68.1 1734.44    72.1 1734.03    84.1 1733.66
   90.591732.209    92.1 1731.88    96.1 1731.72   100.1 1731.72  109.331732.234
   120.1 1733.61   124.1 1735.27   128.1 1737.34   132.1 1738.99   136.1  1739.9
   148.1 1740.71   156.1 1740.66   177.4 1741.02   190.5 1742.05   199.2 1743.28
   212.2  1746.5   226.6 1747.87   251.5 1750.59   273.3 1753.29   280.9 1754.78
#Mann= 3 ,-1,0
       0      .1       0   90.59    .045       0  109.33      .1       0
Bank Sta=90.59,109.33
XS Rating Curve= 0 ,0
Exp/Cntr(USF)=0,0
Exp/Cntr=0.3,0.1

Type RM Length L Ch R = 1 ,9643    ,161.9,161.9,161.9
XS GIS Cut Line= 2
2212339.98825549723181.687565834 2212571.1748177723029.314604381
#Sta/Elev= 30
       0 1745.91    14.6 1745.67    19.4 1744.79    24.2  1742.4    33.8 1736.42
    38.5 1732.41    42.81730.292    43.8 1730.01    46.7 1729.88    52.5 1729.99
   54.061730.286    61.1 1732.29    66.3 1733.12    95.4 1733.82   110.4 1735.73
     120 1736.48   133.3 1736.54   153.5 1737.03   163.1 1736.91     168 1737.06
   175.4 1737.43   182.6 1738.09   191.8 1738.52   196.9 1739.01   204.4  1740.1
   225.4 1743.85   255.3 1749.62   258.9 1750.17     269  1751.1   276.9 1753.06
#Mann= 3 ,-1,0
       0      .1       0    42.8    .045       0   54.06      .1       0
Bank Sta=42.8,54.06
XS Rating Curve= 0 ,0
Exp/Cntr(USF)=0,0
Exp/Cntr=0.3,0.1

Type RM Length L Ch R = 1 ,9481    ,39.1,39.1,39.1
XS GIS Cut Line= 4
 2212393.3886734 723365.335655592212470.60834789723297.768440412
2212551.96479065723162.6340100552212626.42661962 723102.65087005
#Sta/Elev= 30
       0 1744.89     6.3 1745.15    12.4 1744.73    16.3 1743.84    24.8 1742.68
    35.6 1738.17    46.2 1736.67    91.4    1734   103.3 1733.64   112.9 1733.79
     122 1732.83   126.6 1732.03   131.3 1729.92   136.2 1728.37   144.4 1727.92
  147.421728.374   156.6 1730.65   162.5  1731.2   168.7 1731.06     192  1732.2
   238.7 1732.47   243.4  1732.6   252.7  1733.8   260.6 1733.62   264.4 1733.96
   275.4 1736.12   300.9  1743.2   312.7 1745.43     327 1747.62     356 1754.33
#Mann= 3 ,-1,0
       0      .1       0   136.2    .045       0  147.42      .1       0
#XS Ineff= 2 , 0
                          164.77         1734.67
Permanent Ineff=
       F       F
Bank Sta=136.2,147.42
XS Rating Curve= 0 ,0
Exp/Cntr(USF)=0,0
Exp/Cntr=0.3,0.1

Type RM Length L Ch R = 1 ,9442    ,112.6,112.6,112.6
XS GIS Cut Line= 4
2212421.65658995723392.5693800752212498.87626444723325.002164897
2212580.23270721 723189.867734542212654.69453618723129.884594535
#Sta/Elev= 30
       0 1738.66     3.3 1738.29    47.7  1737.7    67.1 1736.07    83.1 1735.53
   102.6 1733.21   116.4 1733.26   125.7 1731.29  134.331727.789   136.1 1727.31
   143.9  1727.1   150.1  1727.8   155.9 1730.09   164.6 1731.81   182.1 1730.94
   195.8 1732.96   199.6 1732.29   205.1 1729.94   208.3 1729.73   214.5 1731.64
   237.5 1731.85   247.1 1733.16   280.6 1735.98   286.9 1737.72   299.7 1743.38
   318.8 1747.96   329.1 1749.93   337.3  1752.2   350.7 1755.05     356 1755.67
#Mann= 3 ,-1,0
       0      .1       0  134.33    .045       0   150.1      .1       0
#XS Ineff= 2 , 0
                          196.69         1735.15
Permanent Ineff=
       F       F
Bank Sta=134.33,150.1
XS Rating Curve= 0 ,0
Exp/Cntr(USF)=0,0
Exp/Cntr=0.3,0.1

Type RM Length L Ch R = 1 ,9329    ,365.6,365.6,365.6
XS GIS Cut Line= 3
2212554.46423264723548.6747960322212636.43037742723273.352617408
2212725.75245827723173.522056456
#Sta/Elev= 30
       0 1744.24    24.5 1739.69    45.4 1736.65    78.2  1729.9    94.2 1727.83
   120.5 1726.33   187.5 1729.56   191.5 1729.32  198.921725.754     204 1725.19
   216.4 1725.75   224.8 1729.01   230.3 1729.84   242.2 1729.25     255 1726.72
   262.4  1726.3   266.6 1727.37   274.3 1730.55   287.3 1731.63   304.9  1729.8
   319.7 1726.45   330.4 1726.32   335.4 1728.19   351.9 1744.16     358 1748.09
   366.5 1750.13   380.7 1750.91   384.1 1751.77   394.8 1757.12   421.2 1761.09
#Mann= 3 ,-1,0
       0      .1       0  198.92    .045       0   216.4      .1       0
#XS Ineff= 2 , 0
          182.07 1733.51  232.93         1733.46
Permanent Ineff=
       F       F
Bank Sta=198.92,216.4
XS Rating Curve= 0 ,0
Exp/Cntr(USF)=0,0
Exp/Cntr=0.3,0.1

Type RM Length L Ch R = 1 ,8964    ,276.2,276.2,276.2
XS GIS Cut Line= 2
2212624.87104931723644.301964943 2212822.4304752 723397.35268259
#Sta/Elev= 30
       0 1746.35     4.6 1746.43     9.1 1745.98    14.2 1744.75    19.4 1742.96
    24.5 1741.66    41.6 1734.32    55.2 1726.29    60.3 1723.69    62.9 1722.81
      70 1722.33    75.7 1722.47   77.781722.829    80.8 1723.57      86 1725.74
    91.1 1726.44   109.9 1726.43   142.3 1727.67   197.4 1728.48   203.8    1729
   216.6 1731.33   234.5 1733.67   248.6 1736.57   257.9 1739.54   263.5  1740.6
   280.6 1740.94   294.8 1741.94   299.8 1743.12   306.2 1745.44   316.2 1747.89
#Mann= 3 ,-1,0
       0      .1       0    62.9    .045       0   77.78      .1       0
Bank Sta=62.9,77.78
XS Rating Curve= 0 ,0
Exp/Cntr(USF)=0,0
Exp/Cntr=0.3,0.1

Type RM Length L Ch R = 1 ,8687    ,385.9,385.9,385.9
XS GIS Cut Line= 2
2212686.98784279723711.322715804  2213023.259206723608.573132603
#Sta/Elev= 30
       0 1743.51     5.9 1741.56    15.5 1740.38    22.2  1737.8    34.7 1734.09
    50.7 1731.17    59.8 1730.07    76.5  1728.4    88.9 1728.17    97.4 1727.42
   147.6 1727.34   181.1 1726.22   185.3 1725.72   189.5 1723.67  192.921721.301
   197.8 1720.37     202 1721.25   218.7 1724.28   260.6 1724.22   265.4 1725.67
   273.1 1729.33   281.5  1732.2   285.7 1734.92   289.8 1738.54   294.8 1741.41
   298.2 1742.14   314.9 1741.58   331.7 1742.26   339.1 1743.29   351.6 1746.44
#Mann= 3 ,-1,0
       0      .1       0  192.92    .045       0     202      .1       0
#XS Ineff= 2 , 0
                          223.98         1726.86
Permanent Ineff=
       F       F
Bank Sta=192.92,202
XS Rating Curve= 0 ,0
Exp/Cntr(USF)=0,0
Exp/Cntr=0.3,0.1

Type RM Length L Ch R = 1 ,8302    ,448.4,453.4,450.1
XS GIS Cut Line= 2
 2212807.2515595723909.816228807 2213024.4268149723833.921650306
#Sta/Elev= 30
       0 1730.91     5.2 1729.58    26.4 1725.44    39.1  1724.7    47.6 1724.52
    51.8 1723.83    56.1  1723.4    77.2 1722.33    82.9 1721.81      86 1721.27
      90 1720.04   97.511716.328    98.4 1715.91   101.7 1715.52   106.9 1715.43
   115.4 1715.71   119.6 1716.35   124.2 1718.08   132.3 1720.02   140.8 1723.46
   148.8 1725.16   153.5  1725.8   174.7  1727.9   191.7 1728.64   204.4 1730.51
   212.8 1730.77   217.1 1731.53   224.2 1734.72   225.6 1735.13   230.1 1735.47
#Mann= 3 ,-1,0
       0      .1       0   97.51    .045       0   119.6      .1       0
Bank Sta=97.51,119.6
XS Rating Curve= 0 ,0
Exp/Cntr(USF)=0,0
Exp/Cntr=0.3,0.1

Type RM Length L Ch R = 1 ,7848    ,149.8,153.7,159.9
XS GIS Cut Line= 2
 2212841.1122176 724144.50561771 2213148.1933583724032.415163309
#Sta/Elev= 30
       0 1736.45    14.3 1734.06    28.8 1731.06    33.1 1729.69    39.3 1725.66
    50.1  1716.1    54.4 1713.77   56.341713.283    62.9 1712.78   72.011713.289
    79.9  1716.7    96.9 1718.51   143.8 1719.92   182.1 1723.39   192.2 1722.86
   211.9 1723.64   233.2 1725.61   241.7 1727.52   257.7 1727.93   267.3 1729.65
   275.8  1732.1     280 1732.68   284.3 1732.55   292.8 1730.79   297.1 1730.94
   301.3 1731.47   305.6 1732.99   309.8 1735.63   314.1 1737.13   326.9  1740.2
#Mann= 3 ,-1,0
       0      .1       0   56.34    .045       0   72.01      .1       0
Bank Sta=56.34,72.01
XS Rating Curve= 0 ,0
Exp/Cntr(USF)=0,0
Exp/Cntr=0.3,0.1

Type RM Length L Ch R = 1 ,7694    ,297.4,298.8,291.3
XS GIS Cut Line= 2
2212864.07519263 724265.807208992213213.06051941724250.239090323
#Sta/Elev= 30
       0 1734.71    12.1 1731.47    36.1  1727.1    48.1 1722.25    68.2 1716.23
    80.2  1715.5    84.2 1714.79   91.211712.009   100.4 1711.47   108.2  1711.5
   112.2 1712.03   116.2 1713.84   120.2 1716.89   124.2 1719.03   132.2 1720.26
   144.2 1720.83     154 1720.49   180.3 1721.09   192.3 1720.06   200.3 1721.81
   208.3 1720.52   212.3 1720.59   260.4 1723.58   272.8 1725.85     292 1728.29
   312.4 1727.24   316.4 1727.45   324.4 1731.06   328.4  1732.2   349.3 1736.31
#Mann= 3 ,-1,0
       0      .1       0   91.21    .045       0   112.2      .1       0
Bank Sta=91.21,112.2
XS Rating Curve= 0 ,0
Exp/Cntr(USF)=0,0
Exp/Cntr=0.3,0.1

Type RM Length L Ch R = 1 ,7396    ,279.3,281.3,272
XS GIS Cut Line= 2
2212892.61674352724482.4635271042213244.19675675724421.488395659
#Sta/Elev= 30
       0 1729.17     7.7 1727.78    15.8 1726.97    23.9 1724.99    60.4 1719.09
    76.7 1716.07    87.2 1714.82      97 1714.79   105.1    1714   125.4  1714.1
     146 1713.59   177.2 1711.72   194.4 1711.59   198.5 1711.03  206.871708.689
   211.8 1708.19   222.8 1708.21  227.481708.672     235 1711.98   243.1  1716.9
   247.2 1718.52   255.3 1719.19   287.9 1718.12     300 1719.12     304 1720.92
   312.1 1726.38   316.2 1727.68   332.4 1731.48   348.7 1733.81   356.8 1735.69
#Mann= 3 ,-1,0
       0      .1       0  206.87    .045       0  227.48      .1       0
Bank Sta=206.87,227.48
XS Rating Curve= 0 ,0
Exp/Cntr(USF)=0,0
Exp/Cntr=0.3,0.1

Type RM Length L Ch R = 1 ,7114    ,246.2,252.3,248.6
XS GIS Cut Line= 2
2212877.04862485724686.1464129962213274.03565086724542.141315327
#Sta/Elev= 30
       0 1734.34     7.6 1732.17    20.3 1730.22    45.9 1724.02    50.1 1720.92
    62.5 1708.23    67.2 1704.77    71.9 1702.44    78.1 1701.75    92.7 1702.46
   101.2 1705.39   105.4 1705.67   126.7 1705.84   152.3 1707.82     165 1706.86
   174.9 1707.53     182 1707.01   186.3 1707.58   194.8 1710.83   207.6 1707.94
     214 1707.45   254.4 1707.41   262.4 1709.06   274.8 1714.28   281.1 1715.33
     365 1717.06   374.8 1718.81   386.3 1724.57   390.5 1725.87   422.3 1732.62
#Mann= 3 ,-1,0
       0      .1       0    71.9    .045       0    92.7      .1       0
Bank Sta=71.9,92.7
XS Rating Curve= 0 ,0
Exp/Cntr(USF)=0,0
Exp/Cntr=0.3,0.1

Type RM Length L Ch R = 1 ,6862    ,189.8,198.1,198.7
XS GIS Cut Line= 2
2212905.59017574724849.6116589982213342.79484164724802.907302998
#Sta/Elev= 30
       0 1729.63     6.6 1728.19    18.7 1726.73    29.4 1723.72    58.9 1718.05
      79 1713.31   119.5 1704.94   146.5 1701.49   159.5 1700.42   167.5 1698.22
   171.6 1697.58   187.6 1698.55   191.7 1698.28  204.841695.886   211.8 1695.31
   218.6 1695.88   227.9  1699.3   231.9 1699.62   260.1 1699.12   272.1 1698.22
   316.4 1697.69   320.4 1698.27   336.5 1702.42   344.5 1703.98   364.6 1706.01
   376.7 1708.88     388 1709.96   400.9 1714.21   417.1 1717.01   439.7 1721.96
#Mann= 3 ,-1,0
       0      .1       0  204.84    .045       0   218.6      .1       0
#XS Ineff= 2 , 0
          182.07 1701.14  239.82         1704.12
Permanent Ineff=
       F       F
Bank Sta=204.84,218.6
XS Rating Curve= 0 ,0
Exp/Cntr(USF)=0,0
Exp/Cntr=0.3,0.1
